--- NFrkAntCk.prj (project) ---

Proj Title=NFrkAntCk
Current Plan=p01
Default Exp/Contr=0,0
English Units
Geom File=g01
Flow File=f01
Plan File=p01
BEGIN DESCRIPTION:
END DESCRIPTION:
DSS Export Rating Curves= 0
DSS Export Rating Curve Sorted= 0
DSS Export Volume Flow Curves= 0
DXF OffsetX= 0
DXF OffsetY= 0
DXF ScaleX= 0
DXF ScaleY= 0

--- NFrkAntCk.p01 (plan) ---

Plan Title=Floodplain
Program Version=4.00
Geom File=g01
Flow File=f01
K Sum by GR=0
Std Step Tol=0.01
Critical Tol=0.01
Num of Std Step Trials=20
Max Error Tol=0.3
Flow Tol Ratio=0.001
Split Flow NTrial=30
Split Flow Tol=0.02
Split Flow Ratio=0.02
Log Output Level=0
Friction Slope Method=1
Unsteady Friction Slope Method=2
Unsteady Bridges Friction Slope Method=1
Global Log Level=0
CheckData=False
Run HTab=0
Run UNet=0
Run PostProcess=0
UNET Theta=0
UNET Theta Warmup=0
UNET ZTol=0
UNET ZSATol=0
UNET MxIter=0
UNET MaxInSteps=0
UNET DtIC=0
UNET DtMin=0
UNET MaxCRTS=0
UNET WFStab=0
UNET SFStab=0
UNET WFX=0
UNET SFX=0
UNET DSS MLevel=0
UNET DZMax Abort=0
UNET Convert EG Bridges=0
UNET Use Existing IB Tables=0
UNET Froude Limit=0
UNET Froude Power=0
Write IC File=0
Echo Input=False
Echo Output=False
Write Detailed=0

--- NFrkAntCk.f01 (steady flow) ---

Flow Title=NFF Regression Equation
Program Version=4.00
Number of Profiles=1
Profile Names=P100yr
River Rch & RM=NFrkAntCk,Main      ,44140.3
1382.934
River Rch & RM=NFrkAntCk,Main      ,41883.8
1413.581
River Rch & RM=NFrkAntCk,Main      ,41538.2
1570.710
River Rch & RM=NFrkAntCk,Main      ,38583.4
1650.121
River Rch & RM=NFrkAntCk,Main      ,35575.5
1825.815
River Rch & RM=NFrkAntCk,Main      ,34182.1
2020.946
River Rch & RM=NFrkAntCk,Main      ,29247.2
2231.582
River Rch & RM=NFrkAntCk,Main      ,24700
2445.771
River Rch & RM=NFrkAntCk,Main      ,19908.5
2707.451
River Rch & RM=NFrkAntCk,Main      ,11710.7
2850.100
River Rch & RM=NFrkAntCk,Main      ,11277.7
3172.359
River Rch & RM=NFrkAntCk,Main      ,8687
3206.484
River Rch & RM=NFrkAntCk,Main      ,37.6
3562.147
Boundary for River Rch & Prof#=NFrkAntCk,Main      ,1
Up Type=0
Dn Type=3
Dn Slope=0.005413

--- NFrkAntCk.g01 (geometry) ---

Geom Title=USGS 10m DEM
Program Version=4.10

River Reach=NFrkAntCk       ,Main
Reach XY= 30
     2233817.084      386383.582     2232379.584      385471.081
     2231887.396      383774.207     2230002.053      382369.375
     2230172.749      381367.729     2229538.114      381043.655
     2228720.185      379751.252     2228762.136      379064.868
     2228052.148      378608.925     2227621.511       376901.42
     2226621.384      376052.012     2226474.018       375123.13
     2224574.636      373156.628     2224728.282       372251.68
     2223935.495      370969.608     2223989.994      370086.789
     2221904.139      368827.501     2220048.594       364564.18
     2218835.052      363685.274     2218507.246      362496.801
     2217465.764      361568.078     2217251.927      360068.969
     2217676.701      359388.391     2217156.389      358452.453
     2217592.327      357750.891     2217132.951      356886.828
     2217517.326      356561.828     2217531.389      355685.266
     2218537.639      354558.703      2218893.36      353277.844

Type RM Length L Ch R = 1 ,44140.3 ,765.6,760.8,758.2
XS GIS Cut Line= 3
     2234234.823      386050.475     2233735.644      386407.756
     2233076.829      386742.231
#Sta/Elev= 30
       0  2566.7    30.2 2558.55    70.4 2550.96    90.6 2548.93   100.6  2546.7
   130.8 2535.86   140.9 2531.14   201.3 2496.82   352.2 2399.37   362.3 2393.86
   372.3 2390.67   382.4 2390.18   462.9 2390.55     495 2387.98   503.2 2387.75
     510 2387.97   573.6 2392.71   703.7 2394.12   873.5  2399.9   993.3 2413.54
  1063.2  2429.2  1103.1 2439.74  1123.1  2447.2    1163 2464.58    1183 2471.48
  1212.9 2480.49  1262.9 2492.34  1292.8 2501.11  1322.8  2512.4  1352.7 2526.39
#Mann= 3 , 0 , 0
       0      .1       0     495    .045       0     510      .1       0
Bank Sta=495,510
XS Rating Curve= 0 ,0
Exp/Cntr=0.3,0.1

Type RM Length L Ch R = 1 ,43379.4 ,323,324.4,325.7
XS GIS Cut Line= 2
     2233551.157       385578.45     2232784.401      386467.571
#Sta/Elev= 30
       0 2517.93    30.1 2506.54    50.2 2497.85   130.4 2460.66   160.6 2445.97
   200.7 2425.36   250.9 2401.39   260.9    2397   270.9 2394.26     281 2392.93
   311.1 2390.38   421.5 2385.32   484.2 2381.38   499.2 2380.98   501.7 2380.97
   531.8  2382.7     572 2383.12   692.4 2381.67   762.6 2382.84     873  2388.9
   923.2 2390.63   933.2 2391.49   943.3 2392.87   973.4 2401.44   993.4    2406
  1003.5 2407.58  1073.7  2405.7  1103.8  2406.2  1123.9 2407.24  1174.1 2407.17
#Mann= 3 , 0 , 0
       0      .1       0   484.2    .045       0   499.2      .1       0
Bank Sta=484.2,499.2
XS Rating Curve= 0 ,0
Exp/Cntr=0.3,0.1

Type RM Length L Ch R = 1 ,43055   ,243.6,245.5,247.4
XS GIS Cut Line= 2
     2233337.783      385374.775      2232552.18      386184.625
#Sta/Elev= 30
       0  2465.2    20.2 2454.99    60.4 2436.73     131 2409.12     141 2405.54
   151.1  2403.2   191.4  2399.8   453.3  2383.6   473.5 2381.87   493.6 2378.72
   499.4 2378.46   503.7 2378.26   514.4 2378.76   533.9 2380.19     544 2380.21
   614.5  2378.8   664.9 2378.76   735.4 2379.59   785.8 2379.35   866.4 2378.17
   876.4 2379.15   886.5 2382.23   896.6 2387.45   916.7 2399.95   926.8 2406.76
     947  2421.6   987.2 2453.55  1017.5 2476.01  1077.9 2517.35  1128.3 2550.66
#Mann= 3 , 0 , 0
       0      .1       0   499.4    .045       0   514.4      .1       0
Bank Sta=499.4,514.4
XS Rating Curve= 0 ,0
Exp/Cntr=0.3,0.1

Type RM Length L Ch R = 1 ,42809.5 ,536.3,544.6,552.9
XS GIS Cut Line= 2
     2233113.966       385311.16      2232342.96      385989.181
#Sta/Elev= 30
       0 2400.12    60.4 2395.83   171.1 2386.09   211.4 2383.16   241.6 2381.51
   281.8 2379.93     302  2379.5   322.1 2379.74   332.2 2379.52   354.4 2378.09
   369.4 2378.51   392.6  2379.8   402.6 2379.84   563.7 2376.63   624.1  2376.4
   654.3 2376.73   704.6 2374.78   714.7 2374.93   724.8 2377.16   734.8 2382.62
   744.9 2389.54   775.1 2411.28   845.5 2463.97   905.9 2508.04     916 2514.65
   926.1 2519.52   936.1 2520.86   946.2 2520.52   976.4 2518.53  1026.7 2516.17
#Mann= 3 , 0 , 0
       0      .1       0   354.4    .045       0   369.4      .1       0
Bank Sta=354.4,369.4
XS Rating Curve= 0 ,0
Exp/Cntr=0.3,0.1

Type RM Length L Ch R = 1 ,42264.6 ,385,380.2,375.3
XS GIS Cut Line= 3
     2233095.313       385253.54      2232634.62      385326.281
     2232125.433      385539.655
#Sta/Elev= 30
       0  2399.7   148.8 2389.98   168.7 2388.86   198.5 2387.52   307.6 2384.45
   436.6  2381.2   476.4  2379.5   526.6 2377.71   556.7 2377.06   596.9 2376.57
   667.2 2374.62   727.4 2373.64   759.6 2372.38   774.6 2371.61   777.6 2371.49
   787.6 2372.21   797.6 2375.67   807.7  2380.7   827.8 2389.86   837.8 2394.64
   847.8 2399.95   857.9  2405.9     878 2419.13   918.1 2447.07   928.2 2453.88
   938.2 2460.26   948.2 2465.42   958.3 2468.38   968.3 2469.57  1018.5 2471.58
#Mann= 3 , 0 , 0
       0      .1       0   759.6    .045       0   774.6      .1       0
Bank Sta=759.6,774.6
XS Rating Curve= 0 ,0
Exp/Cntr=0.3,0.1

Type RM Length L Ch R = 1 ,41883.8 ,345.7,345.7,345.7
XS GIS Cut Line= 2
     2232784.952      384749.202     2232018.746       385253.54
#Sta/Elev= 30
       0 2403.31    20.2 2401.67    60.5 2398.95   181.4 2391.43   191.5 2390.54
   201.6 2389.15   221.8  2385.3   231.8 2384.07     252 2382.75   342.7 2378.84
   433.4 2373.94   483.8 2371.87     504 2371.38   604.8 2370.84   638.7  2368.9
   645.1 2368.84   653.7 2369.28   725.8 2374.19   735.8 2375.48   745.9 2378.08
     756 2381.71   766.1 2385.86   776.2  2390.4   796.3 2400.42   826.6 2416.76
     877 2445.53     887 2450.51   897.1 2453.54   907.2 2455.82   917.3  2456.9
#Mann= 3 , 0 , 0
       0      .1       0   638.7    .045       0   653.7      .1       0
Bank Sta=638.7,653.7
XS Rating Curve= 0 ,0
Exp/Cntr=0.3,0.1

Type RM Length L Ch R = 1 ,41538.2 ,818.4,816.9,814
XS GIS Cut Line= 2
     2232581.277      384482.485     2231829.619      384972.275
#Sta/Elev= 30
       0 2390.94     121 2379.83   151.2 2376.04   171.4 2374.42   302.4 2371.14
   332.6 2368.51   362.9 2368.84   453.6 2368.13   524.2 2368.44     625 2370.15
   645.1 2369.98   671.5 2368.88   686.5 2368.72   695.6  2369.8   715.7 2374.96
   735.9 2381.77     746 2385.89     756 2390.84   766.1 2396.75   776.2 2403.88
   786.3  2412.2   796.4 2421.72   826.6 2451.67   836.7 2459.91   846.8 2466.46
   856.8 2471.35   866.9 2474.71     877 2477.11   887.1 2478.65   897.2 2479.16
#Mann= 3 , 0 , 0
       0      .1       0   671.5    .045       0   686.5      .1       0
Bank Sta=671.5,686.5
XS Rating Curve= 0 ,0
Exp/Cntr=0.3,0.1

Type RM Length L Ch R = 1 ,40721.3 ,594.3,593.1,593.2
XS GIS Cut Line= 2
     2232348.505      383973.298      2231577.45      384574.624
#Sta/Elev= 30
       0 2398.66    40.3  2394.5   100.8 2389.57   262.1 2380.08   282.3 2378.59
   332.7 2372.38   342.7 2370.79   383.1 2362.38   393.1 2361.11     410  2360.4
     425 2361.02   443.5 2362.98   453.6  2363.3   544.4 2360.97   614.9 2360.05
   645.2  2360.4   725.8 2362.54   766.1 2362.56   776.2 2363.49   786.3 2366.61
   796.4 2371.46   806.4 2376.88   826.6 2388.64   856.8 2407.78   927.4 2454.51
   937.5 2460.96   947.6 2466.96   957.6 2470.37   967.7 2471.05   977.8 2470.88
#Mann= 3 , 0 , 0
       0      .1       0     410    .045       0     425      .1       0
Bank Sta=410,425
XS Rating Curve= 0 ,0
Exp/Cntr=0.3,0.1

Type RM Length L Ch R = 1 ,40128.2 ,762.9,753.8,744.7
XS GIS Cut Line= 2
     2232115.734      383488.358     2231242.271      384151.063
#Sta/Elev= 30
       0 2472.44    50.3 2447.64   100.6 2424.16   110.6 2420.19   120.7 2417.11
   160.9    2408   221.3 2388.41   301.8 2368.75   331.9 2358.38   352.1 2353.01
   359.5 2351.81   374.5 2351.19   382.2 2351.91   402.4  2356.9   412.4 2356.01
   432.5 2351.76   442.6 2350.75   502.9  2349.6   824.8 2351.74     855 2352.69
   865.1  2355.3   885.2 2364.14   915.4 2378.76   935.5 2389.84   955.6 2401.84
   985.8 2421.39  1036.1 2456.89  1066.2 2477.06  1086.4 2489.72  1096.4 2494.07
#Mann= 3 , 0 , 0
       0      .1       0   359.5    .045       0   374.5      .1       0
Bank Sta=359.5,374.5
XS Rating Curve= 0 ,0
Exp/Cntr=0.3,0.1

Type RM Length L Ch R = 1 ,39374.4 ,783,791,799
XS GIS Cut Line= 2
     2231548.853      382720.067     2230863.917      383927.043
#Sta/Elev= 30
       0 2474.68    50.3 2459.26   130.7 2431.58   201.1 2413.11   231.3 2406.19
   301.7 2393.24     362 2380.72   432.4 2367.19   492.8 2351.25   512.9 2349.28
   593.3 2344.89   719.7 2341.79   734.1 2341.57   734.7 2341.59   874.9 2349.18
   955.4 2352.06   975.5 2353.61  1005.6 2359.36  1116.3 2378.07  1126.3  2380.5
  1136.4 2383.98  1216.8 2416.97  1236.9 2426.37  1287.2 2451.96  1307.3 2460.65
  1317.4 2463.35  1327.4  2464.8  1337.5 2465.03  1357.6  2463.3  1387.8 2456.62
#Mann= 3 , 0 , 0
       0      .1       0   719.7    .045       0   734.7      .1       0
Bank Sta=719.7,734.7
XS Rating Curve= 0 ,0
Exp/Cntr=0.3,0.1

Type RM Length L Ch R = 1 ,38583.4 ,773.7,781.3,788.9
XS GIS Cut Line= 2
     2231102.209      382474.833     2230195.371      383255.586
#Sta/Elev= 30
       0 2452.24    60.3 2441.08   140.8 2428.93     181 2424.07   191.1 2421.64
   211.2 2414.48   251.4 2397.67   301.7 2375.13   372.1 2349.32   382.1  2346.7
   402.2    2345     543 2336.99   603.3 2334.59   610.3 2334.62   625.3 2335.36
   653.6 2336.67   764.2 2338.38   784.4  2340.1   824.6  2345.6   844.7 2347.62
   884.9 2350.31   945.2 2353.25   955.3 2354.69   995.5  2367.5  1035.7 2375.64
  1045.8 2379.07  1156.4 2427.84  1166.5 2431.05  1176.5 2432.08  1196.6 2431.56
#Mann= 3 , 0 , 0
       0      .1       0   610.3    .045       0   625.3      .1       0
Bank Sta=610.3,625.3
XS Rating Curve= 0 ,0
Exp/Cntr=0.3,0.1

Type RM Length L Ch R = 1 ,37801.7 ,787.1,792.1,797.1
XS GIS Cut Line= 2
     2230748.183       382088.84     2229579.497      382615.465
#Sta/Elev= 30
       0 2445.89    60.6 2440.13    90.8 2433.67   151.4 2408.41   282.6 2366.62
   333.1 2348.96   373.4 2333.32   383.6 2331.28   615.7 2328.41   726.7 2328.98
   767.1 2328.12   771.2 2328.43   786.2  2329.9   837.8 2331.22   847.8 2332.72
   857.9  2337.7   878.1 2356.44   888.2 2363.45   898.3 2366.55   918.5 2370.44
   928.6 2375.44   999.2 2419.52  1009.3 2424.46  1029.5 2431.74  1049.7 2437.25
  1140.6 2453.54  1201.1  2467.6  1221.3 2475.06  1261.7 2493.56  1281.9  2503.9
#Mann= 3 , 0 , 0
       0      .1       0   771.2    .045       0   786.2      .1       0
Bank Sta=771.2,786.2
XS Rating Curve= 0 ,0
Exp/Cntr=0.3,0.1

Type RM Length L Ch R = 1 ,37009.5 ,837.4,824.4,811.4
XS GIS Cut Line= 2
     2230723.956      381572.844     2229356.552      381748.135
#Sta/Elev= 30
       0 2491.87   110.7 2442.84   201.2 2409.19   271.7 2371.14   291.8  2361.3
   382.4 2326.09   392.4 2323.32   412.6 2322.25   593.7 2323.36   617.7  2321.5
   632.7 2320.42     634 2320.36   674.2 2322.57   835.2 2321.92   976.1 2324.69
   986.2  2326.1  1006.3 2332.34  1056.6 2355.66  1066.6 2358.16  1076.7 2358.75
  1137.1 2352.77  1167.3  2347.5  1177.3 2346.58  1187.4 2347.36  1197.5 2350.03
  1207.5 2354.63  1237.7 2372.35  1328.3 2422.05  1348.4 2431.57  1378.6 2443.57
#Mann= 3 , 0 , 0
       0      .1       0   617.7    .045       0   632.7      .1       0
Bank Sta=617.7,632.7
XS Rating Curve= 0 ,0
Exp/Cntr=0.3,0.1

Type RM Length L Ch R = 1 ,36185.1 ,608.7,609.6,610.2
XS GIS Cut Line= 2
      2230200.22      380670.855     2229275.554       381583.63
#Sta/Elev= 30
       0 2516.25    30.2 2494.22    60.4  2474.5   110.8 2443.32   151.1 2420.16
   171.2 2409.62   191.4 2400.67   251.8 2378.62   372.7 2347.15   433.1 2327.82
   473.4 2316.68   493.5 2314.37   584.2  2314.2   632.8 2310.41   634.5  2310.3
   647.8 2310.34   674.8 2311.57   775.6    2320   805.8 2320.91   866.2 2320.18
   926.6 2322.94   936.7 2323.87   966.9 2330.89   987.1 2338.71  1178.4 2432.14
  1218.7 2455.72  1228.8 2460.38  1238.9 2464.04  1269.1 2471.11  1299.3 2474.41
#Mann= 3 , 0 , 0
       0      .1       0   632.8    .045       0   647.8      .1       0
Bank Sta=632.8,647.8
XS Rating Curve= 0 ,0
Exp/Cntr=0.3,0.1

Type RM Length L Ch R = 1 ,35575.5 ,865.6,865.1,864.6
XS GIS Cut Line= 2
     2229916.351      380330.866     2228799.347      381172.865
#Sta/Elev= 30
       0 2562.69    20.1 2549.64    50.3  2527.8   100.6 2494.63   140.9 2470.51
     312 2373.39   362.3 2341.92   392.5 2319.69   402.5 2315.66   412.6 2314.19
   442.8 2312.71   623.9 2309.49     634 2309.22   647.3  2307.4   662.3 2305.66
   664.2 2305.51   855.4 2315.17   925.8 2322.25   986.2 2329.84  1096.9 2341.12
    1107 2342.87    1117 2346.14  1127.1 2350.67  1157.3 2365.07  1217.7 2392.06
    1278 2420.72  1288.1 2424.38  1308.2 2427.51  1358.6 2429.85  1398.8 2435.75
#Mann= 3 , 0 , 0
       0      .1       0   647.3    .045       0   662.3      .1       0
Bank Sta=647.3,662.3
XS Rating Curve= 0 ,0
Exp/Cntr=0.3,0.1

Type RM Length L Ch R = 1 ,34710.4 ,518.5,528.2,538
XS GIS Cut Line= 2
     2229414.617      379700.975     2228454.436      380438.084
#Sta/Elev= 30
       0 2421.35    50.4 2402.68    80.7 2396.66   100.9 2391.28   141.2 2373.01
   181.6 2357.59     232 2341.37   282.4 2327.23   302.6 2324.27   332.9 2323.33
   423.7 2315.41   518.3 2300.52   524.5 2300.38   533.3  2301.5   554.8 2307.31
   564.9 2308.46   655.7 2302.89   776.7 2304.93   796.9 2307.27   817.1 2313.85
   837.2 2318.25   897.8 2324.54   948.2 2332.33   978.5 2333.57   998.6 2340.36
  1028.9 2354.56  1049.1 2361.94  1069.3 2367.92  1129.8 2381.41  1210.5  2412.7
#Mann= 3 , 0 , 0
       0      .1       0   518.3    .045       0   533.3      .1       0
Bank Sta=518.3,533.3
XS Rating Curve= 0 ,0
Exp/Cntr=0.3,0.1

Type RM Length L Ch R = 1 ,34182.1 ,492.9,484.7,472.7
XS GIS Cut Line= 2
     2229303.081      379477.902      2228095.58      379749.469
#Sta/Elev= 30
       0 2433.31    50.3 2403.11    70.4  2387.1   130.8 2356.19   140.9 2349.64
   150.9 2340.62   171.1 2329.57   191.2 2319.32   201.2 2315.24   211.3 2312.19
   221.4 2308.41   231.4 2307.85   362.2 2307.82   462.9 2305.13     632 2299.47
   633.9 2299.45     647 2299.56   694.3 2300.31   704.4 2300.96   714.4 2302.51
   784.9 2315.97   915.7 2330.68  1016.3 2343.64  1026.4 2346.39  1056.5 2359.18
  1076.7 2368.38    1127  2393.4  1177.3 2415.02  1197.4 2422.76  1237.7 2435.32
#Mann= 3 , 0 , 0
       0      .1       0     632    .045       0     647      .1       0
Bank Sta=632,647
XS Rating Curve= 0 ,0
Exp/Cntr=0.3,0.1

Type RM Length L Ch R = 1 ,33697.5 ,597.7,599.5,608.1
XS GIS Cut Line= 2
     2229181.846      378959.016     2228017.989      379584.589
#Sta/Elev= 30
       0 2466.31    30.3  2458.7    50.4 2449.13    60.5 2439.94     111  2411.1
     121 2405.45   141.2  2397.6   151.3 2385.86   221.9  2347.2     232 2338.27
   262.2 2322.17   282.4 2313.21   322.8 2307.02   373.2 2301.98   413.5 2298.45
   442.6 2298.08   457.6 2298.17   847.3  2300.2   968.3 2297.55   988.5 2299.47
  1018.7 2309.01  1038.9 2318.61  1089.3 2338.47  1109.5  2347.9  1129.7 2360.32
  1149.9 2367.99  1200.3 2393.92  1220.5 2406.34  1230.6 2410.53  1321.3 2460.22
#Mann= 3 , 0 , 0
       0      .1       0   442.6    .045       0   457.6      .1       0
Bank Sta=442.6,457.6
XS Rating Curve= 0 ,0
Exp/Cntr=0.3,0.1

Type RM Length L Ch R = 1 ,33097.9 ,533.6,531.5,526.4
XS GIS Cut Line= 2
     2228813.291      378532.269     2227809.465      379128.745
#Sta/Elev= 30
       0 2430.62    10.1 2427.95    30.2 2419.37    60.4 2411.35   100.7 2395.38
   120.8  2383.5   191.3 2350.36   211.4 2337.64   251.6 2319.64   281.8 2310.54
   322.1 2308.46   352.3 2299.85   372.4 2295.97   507.9 2292.51   513.4 2292.44
   522.9 2292.48   744.9 2296.72   885.8 2294.36     906 2296.44   926.1 2307.16
   936.2 2316.74   946.2 2323.34   976.4 2335.93  1016.7 2348.33  1036.8 2360.84
  1046.9 2364.82  1107.3 2383.54  1117.3 2387.98  1127.4 2395.12  1167.7 2415.45
#Mann= 3 , 0 , 0
       0      .1       0   507.9    .045       0   522.9      .1       0
Bank Sta=507.9,522.9
XS Rating Curve= 0 ,0
Exp/Cntr=0.3,0.1

Type RM Length L Ch R = 1 ,32566.4 ,443.5,452.3,461.1
XS GIS Cut Line= 2
     2228619.315      378086.124     2227421.513      378828.082
#Sta/Elev= 30
       0 2438.13    10.1 2433.51    20.1 2426.52   120.8 2384.81   301.9 2337.98
   392.5 2326.55   503.2 2319.67   573.7 2309.25   654.2 2306.61   724.6 2287.82
   735.9 2286.65   750.9 2288.09   795.1  2292.4   895.7 2287.68  1026.5 2286.36
  1036.6 2286.44  1046.7 2289.67  1056.7 2295.17  1117.1 2315.82  1137.2 2329.12
  1177.5 2350.99  1217.8  2375.5  1237.9 2391.98    1258 2404.22  1268.1 2410.07
  1288.2 2417.94  1298.3 2424.34  1318.4 2442.11  1388.8 2488.59    1409 2505.64
#Mann= 3 , 0 , 0
       0      .1       0   735.9    .045       0   750.9      .1       0
Bank Sta=735.9,750.9
XS Rating Curve= 0 ,0
Exp/Cntr=0.3,0.1

Type RM Length L Ch R = 1 ,32114   ,304.4,299.7,295
XS GIS Cut Line= 2
     2228444.737      377960.039     2227314.826      378154.016
#Sta/Elev= 30
       0 2378.51    40.2 2368.51    60.3 2361.33   120.7 2346.32   140.8 2338.93
   211.2  2322.6     362 2304.45   412.3 2299.86   432.4 2294.34   442.5 2287.69
   452.5 2285.53   653.7 2281.07   660.4 2281.33   675.4 2283.05   744.2 2289.08
   854.8 2283.22   864.9 2283.03   874.9 2284.78     885 2289.66     895 2296.45
   905.1  2308.5   975.5 2352.01   985.5 2360.29  1045.9 2391.19  1055.9 2400.16
    1066 2406.76  1096.2 2421.21  1116.3 2427.42  1126.3  2427.5  1146.4 2421.83
#Mann= 3 , 0 , 0
       0      .1       0   660.4    .045       0   675.4      .1       0
Bank Sta=660.4,675.4
XS Rating Curve= 0 ,0
Exp/Cntr=0.3,0.1

Type RM Length L Ch R = 1 ,31814.5 ,487.3,485.6,483.9
XS GIS Cut Line= 2
     2228449.586      377523.593      2227368.17      377921.244
#Sta/Elev= 30
       0 2420.27      20 2413.78    30.1 2407.92    90.2 2390.99   110.2 2383.35
   140.3 2375.43   180.4 2366.79   190.4 2362.34   260.5 2342.95   280.5 2333.78
   300.6 2326.93   340.6 2321.04   360.7 2316.58   440.8  2302.7   450.9 2299.93
   470.9 2287.06   480.9 2282.91   490.9 2281.71   571.1 2280.03   741.4 2278.04
   744.9 2278.06   759.9 2278.22   791.5 2278.56   921.8 2283.77   981.9 2282.42
   991.9 2284.88  1011.9 2297.01  1082.1 2321.84  1102.1 2332.56  1152.2 2352.58
#Mann= 3 , 0 , 0
       0      .1       0   744.9    .045       0   759.9      .1       0
Bank Sta=744.9,759.9
XS Rating Curve= 0 ,0
Exp/Cntr=0.3,0.1

Type RM Length L Ch R = 1 ,31328.6 ,337.4,336.4,336.9
XS GIS Cut Line= 2
     2228367.146      377009.557     2227106.302      377610.883
#Sta/Elev= 30
       0 2463.34    60.3  2445.3   130.6 2426.63   140.7 2421.24   150.7 2418.38
   221.1 2401.72   231.1 2396.57   271.3 2387.14   301.5 2378.38   321.6 2370.08
   341.7 2365.05   542.7 2331.72   562.8 2325.05   582.9 2313.39     603 2303.93
     613 2294.82   623.1 2282.51   633.1 2275.22   653.2 2273.98   667.1 2274.21
   682.1  2274.9   844.2 2278.34  1075.3  2278.5  1175.8 2281.89  1195.9 2287.51
  1256.2 2314.24  1276.3 2327.55  1336.6 2359.52  1356.7 2373.29  1396.9 2394.33
#Mann= 3 , 0 , 0
       0      .1       0   667.1    .045       0   682.1      .1       0
Bank Sta=667.1,682.1
XS Rating Curve= 0 ,0
Exp/Cntr=0.3,0.1

Type RM Length L Ch R = 1 ,30992.2 ,610.7,607.2,602.2
XS GIS Cut Line= 3
     2228258.797       376643.59     2227664.174      376977.414
     2227040.347      377262.267
#Sta/Elev= 30
       0 2510.34    50.1 2488.12    80.2 2469.84   150.4 2443.41   180.5 2430.52
   200.6 2428.06   220.6 2422.14   250.7 2416.19     351 2385.11   381.1 2377.37
   431.2 2354.44   451.3 2352.85   521.5 2321.92   541.5 2315.04   561.6 2311.06
   601.7 2307.78   651.8  2278.8   661.9 2274.23   680.4  2271.1     692 2270.53
   695.4 2270.64   823.1 2273.91  1135.8  2276.4  1236.6 2274.05  1256.8 2278.84
  1266.8 2284.54    1287 2291.84  1307.2 2302.67  1327.4 2306.91  1367.7 2311.77
#Mann= 3 , 0 , 0
       0      .1       0   680.4    .045       0   695.4      .1       0
#XS Ineff= 2 , 0
                         1144.35         2276.47
Permanent Ineff=
       F       F
Bank Sta=680.4,695.4
XS Rating Curve= 0 ,0
Exp/Cntr=0.3,0.1

Type RM Length L Ch R = 1 ,30385   ,743.4,742.3,741.3
XS GIS Cut Line= 2
     2227581.543      376282.146      2226718.35      376936.816
#Sta/Elev= 30
       0 2457.67      10 2452.63    20.1  2449.2    30.1 2443.96    40.1 2436.94
   120.4  2396.1   140.4 2381.86   160.5 2370.11   190.6 2351.17   200.6  2346.1
   210.7 2342.65   220.7 2336.66   230.7 2328.48   240.8    2319   280.9 2291.38
   300.9 2278.77     311  2273.3     321 2270.18   341.1 2267.93     350 2267.64
   361.1 2267.57     365 2267.61   772.4 2273.59   942.9 2282.41     953  2283.7
     963  2286.4  1023.2 2307.35  1033.2 2312.64  1063.3  2325.5  1083.4 2335.41
#Mann= 3 , 0 , 0
       0      .1       0     350    .045       0     365      .1       0
Bank Sta=350,365
XS Rating Curve= 0 ,0
Exp/Cntr=0.3,0.1

Type RM Length L Ch R = 1 ,29642.7 ,385.3,395.5,405.7
XS GIS Cut Line= 3
     2227499.103      375966.935     2226868.681      375962.086
     2226209.162      376514.918
#Sta/Elev= 30
       0 2519.49   130.1 2474.16   210.2 2429.48   220.2 2420.67   290.2 2393.09
   300.2 2386.95   360.2 2368.87   370.3 2362.26   430.3 2337.54   440.3 2328.69
   460.3 2319.56   480.3 2312.45   510.4 2305.16   560.4 2277.09   570.4 2273.18
   580.4 2271.26   620.4 2270.13   680.5 2265.33     869 2258.11   870.6 2258.04
     884 2258.53  1000.7  2268.6  1200.8 2275.04  1290.9 2314.88  1310.9 2322.23
    1411 2374.25    1421 2381.73    1441 2392.18    1471 2403.57    1491 2407.24
#Mann= 3 , 0 , 0
       0      .1       0     869    .045       0     884      .1       0
Bank Sta=869,884
XS Rating Curve= 0 ,0
Exp/Cntr=0.3,0.1

Type RM Length L Ch R = 1 ,29247.2 ,949.8,944.4,939
XS GIS Cut Line= 3
     2227062.657      375317.115     2226907.476      375680.821
     2225816.361      375957.236
#Sta/Elev= 30
       0 2472.32    59.3 2456.01   118.6 2423.08   138.4 2414.95   227.4 2388.41
   296.6 2372.88   365.8 2351.02   395.4 2344.36   445.7 2322.97   465.8 2310.63
     516 2289.63   536.1 2276.94   576.3 2260.41   596.4 2257.06   837.6 2254.82
   841.1 2254.88   856.1 2255.64   938.1 2260.22   998.4 2259.42  1018.5 2262.81
  1068.8 2278.09  1149.2 2308.65  1169.3 2320.25  1209.5 2336.24  1239.6 2346.24
    1310 2363.09  1330.1  2371.1  1390.4 2384.29  1460.7 2407.22    1521 2430.12
#Mann= 3 , 0 , 0
       0      .1       0   841.1    .045       0   856.1      .1       0
Bank Sta=841.1,856.1
XS Rating Curve= 0 ,0
Exp/Cntr=0.3,0.1

Type RM Length L Ch R = 1 ,28302.8 ,626.8,625.3,623.9
XS GIS Cut Line= 2
     2226820.187      374667.296     2225709.674      375249.224
#Sta/Elev= 30
       0 2508.68    20.1 2499.89    40.1  2487.1    60.2 2480.83   110.3  2453.8
   130.4 2438.85   210.6 2391.23   220.7 2381.93   270.8 2353.24   300.9 2343.53
     321 2330.75   381.1 2302.58   391.2 2295.82   451.4 2270.93   471.4 2260.28
   481.4 2252.39   501.5 2247.99   611.8 2245.04   615.8 2245.18   630.8 2246.06
   842.5 2253.79   852.6 2255.75   912.7 2288.32   932.8 2303.59  1023.1 2350.58
  1083.2 2368.73  1103.3 2378.04  1173.5 2392.78  1193.6 2401.17  1253.8 2409.83
#Mann= 3 , 0 , 0
       0      .1       0   615.8    .045       0   630.8      .1       0
Bank Sta=615.8,630.8
XS Rating Curve= 0 ,0
Exp/Cntr=0.3,0.1

Type RM Length L Ch R = 1 ,27677.9 ,732.3,732.9,733.6
XS GIS Cut Line= 2
     2226301.301      374211.452     2225365.367      374841.874
#Sta/Elev= 30
       0 2476.51    50.4 2439.75    70.5 2429.03    80.6 2421.52   100.8 2398.74
   110.8 2390.61   120.9 2382.53   161.2 2355.46   181.4 2339.96   201.5 2303.95
   211.6 2288.82   221.7 2278.65   231.7 2271.28   241.8 2266.26     272 2257.11
   332.5 2245.01     534 2243.33   574.3 2239.34   579.9 2239.64   594.9 2241.42
   644.8 2251.32     665 2253.52   705.3 2262.91   866.5 2286.65   947.1 2318.94
   967.2  2330.4  1007.6 2347.13  1037.8 2359.17    1068 2368.89  1128.4 2392.97
#Mann= 3 , 0 , 0
       0      .1       0   579.9    .045       0   594.9      .1       0
Bank Sta=579.9,594.9
XS Rating Curve= 0 ,0
Exp/Cntr=0.3,0.1

Type RM Length L Ch R = 1 ,26944.5 ,559.4,558.1,556.8
XS GIS Cut Line= 2
     2225918.198      373697.415     2225045.306      374172.657
#Sta/Elev= 30
       0 2412.16    20.1 2401.16    40.2 2385.44   110.4 2348.38   130.5  2333.3
   210.8 2293.27   220.9 2286.21   281.1 2255.95   291.1 2249.77   301.2  2240.9
   311.2 2237.41   331.3 2236.76     512 2239.02     590 2232.84   602.4 2232.04
     605 2232.06   622.4 2233.89   652.6 2245.33   682.7  2249.6   712.8 2258.54
   732.9 2267.53   752.9 2280.16   823.2 2312.13   843.3 2326.32   913.6  2364.1
   933.6 2377.46   943.7 2381.21   953.7 2388.22   963.8 2392.25   993.9 2408.46
#Mann= 3 , 0 , 0
       0      .1       0     590    .045       0     605      .1       0
Bank Sta=590,605
XS Rating Curve= 0 ,0
Exp/Cntr=0.3,0.1

Type RM Length L Ch R = 1 ,26386.5 ,640,644.4,648.8
XS GIS Cut Line= 2
     2225680.578      373183.379     2224822.234      373702.265
#Sta/Elev= 30
       0  2401.2    70.2  2362.9   150.4 2325.29   160.5 2317.67   220.7 2291.16
   230.7 2285.65   240.7 2274.72   260.8 2259.45   280.8 2249.67   290.9 2241.48
   310.9 2235.64     331 2233.68   481.4 2230.62   611.8  2231.5     682 2227.38
     697 2227.93   732.2 2229.53   742.2 2231.57   752.2 2236.24   782.3 2254.99
   802.4 2272.31   872.6  2317.8   882.6 2325.15   892.7 2334.92   922.8 2353.31
   942.8  2362.9   952.8  2370.5   972.9 2378.62   982.9 2385.54    1003 2394.16
#Mann= 3 , 0 , 0
       0      .1       0     682    .045       0     697      .1       0
Bank Sta=682,697
XS Rating Curve= 0 ,0
Exp/Cntr=0.3,0.1

Type RM Length L Ch R = 1 ,25741.9 ,373.5,381.2,388.8
XS GIS Cut Line= 3
     2225646.632      373076.692     2225059.854      373037.897
     2224235.456      373338.559
#Sta/Elev= 30
       0 2394.77    19.9  2384.2    69.8 2367.16    89.7 2357.84   139.5 2344.04
   169.4 2332.67   249.2 2310.47   378.8 2281.05   428.6 2256.75   458.5 2245.11
   528.3 2236.23   608.2 2244.72   648.6 2245.18   729.3 2229.71   769.6 2229.99
   890.6 2222.48  1066.4 2220.54  1072.2 2220.39  1081.4 2220.47  1092.4 2222.49
  1112.6 2237.59    1163 2263.12  1193.2 2290.01  1253.8 2334.87  1273.9 2355.31
  1314.3 2381.35  1354.6  2402.6  1415.1 2422.46  1425.2 2430.22  1465.6 2450.55
#Mann= 3 , 0 , 0
       0      .1       0  1066.4    .045       0  1081.4      .1       0
Bank Sta=1066.4,1081.4
XS Rating Curve= 0 ,0
Exp/Cntr=0.3,0.1

Type RM Length L Ch R = 1 ,25360.5 ,663.7,660.7,657.7
XS GIS Cut Line= 3
     2225287.776      372485.065     2224996.812      372829.372
     2224182.112       372843.92
#Sta/Elev= 30
       0 2382.22      30 2373.87   100.2 2362.28   110.2 2358.78   200.4 2314.64
   220.4 2302.95   320.6 2265.29   340.6 2254.12   370.6 2242.68   390.7  2240.4
   531.3 2236.88   591.6 2221.67   682.2 2223.54     818 2216.53     823 2216.32
     833 2216.34   863.2 2220.18   903.5 2237.34   913.5 2247.49     984 2289.95
     994 2302.03  1004.1 2309.12  1054.4 2338.15  1064.4 2348.91  1134.8 2385.66
  1144.9 2394.74    1165 2404.68  1205.3 2418.82  1215.3 2424.68  1265.6 2440.19
#Mann= 3 , 0 , 0
       0      .1       0     818    .045       0     833      .1       0
Bank Sta=818,833
XS Rating Curve= 0 ,0
Exp/Cntr=0.3,0.1

Type RM Length L Ch R = 1 ,24700   ,724,710.5,697.1
XS GIS Cut Line= 2
      2225176.24      372131.058     2224094.823      372300.787
#Sta/Elev= 30
       0 2404.82    50.2 2375.88    60.3 2368.73    70.3 2358.66   130.6 2323.14
   140.6 2312.54   210.9  2270.5   220.9 2258.25   291.2 2211.31   301.3 2210.08
   331.4 2210.07   464.2 2210.68   479.2 2211.22   562.4 2216.07   652.8  2216.2
   662.8 2217.15   682.9  2223.1     693 2224.58   743.2 2229.28   773.3 2247.83
   823.5 2269.71   833.5 2276.78   893.8 2300.82   903.8 2309.34   913.9 2314.36
     944 2323.05   964.1 2327.48  1034.4  2332.5  1064.5 2338.59  1094.7 2346.41
#Mann= 3 , 0 , 0
       0      .1       0   464.2    .045       0   479.2      .1       0
Bank Sta=464.2,479.2
XS Rating Curve= 0 ,0
Exp/Cntr=0.3,0.1

Type RM Length L Ch R = 1 ,23989.4 ,563.8,580.2,596.6
XS GIS Cut Line= 2
      2224773.74      371233.919     2223871.751      372058.317
#Sta/Elev= 30
       0 2432.37      30 2422.16    60.1 2408.13   140.2 2386.94   250.4 2341.25
   270.4  2329.3   290.5 2320.15   310.5 2313.76   360.6 2288.24   380.6 2272.96
   390.6 2267.22   440.7 2240.43   460.7 2234.17   480.8 2220.19   490.8 2210.16
   500.8    2204     507 2202.78   510.8 2202.04     522 2202.37     611 2208.46
   791.3 2210.31   841.4 2215.44   891.4 2229.21   961.6 2239.57  1021.6 2258.52
  1041.7  2265.2  1081.8 2282.58  1101.8 2287.95  1161.9 2316.31    1222 2338.86
#Mann= 3 , 0 , 0
       0      .1       0     507    .045       0     522      .1       0
Bank Sta=507,522
XS Rating Curve= 0 ,0
Exp/Cntr=0.3,0.1

Type RM Length L Ch R = 1 ,23409.3 ,431.6,428.9,426.1
XS GIS Cut Line= 2
     2224652.504      371107.835     2223537.142      371170.877
#Sta/Elev= 30
       0 2357.57    40.3 2341.66    60.4 2330.26   120.8 2308.67   130.8 2302.54
   201.3 2279.55   211.4 2273.83   281.8 2252.44   342.2 2239.46   362.3 2231.42
   503.2 2206.25   513.3 2202.29   613.9 2200.79   625.7 2200.85   640.7 2201.07
   704.5 2202.24   724.6 2207.44   734.7 2223.12   754.8 2244.54     775  2258.6
   805.2 2275.66   815.2 2284.24   875.6 2311.66   885.7 2319.13   915.9 2330.33
   976.2 2359.67  1026.6  2374.9  1046.7 2383.23    1097 2399.16  1117.1 2410.45
#Mann= 3 , 0 , 0
       0      .1       0   625.7    .045       0   640.7      .1       0
Bank Sta=625.7,640.7
XS Rating Curve= 0 ,0
Exp/Cntr=0.3,0.1

Type RM Length L Ch R = 1 ,22980.3 ,699,690.6,680.1
XS GIS Cut Line= 2
     2224667.053       370656.84     2223415.907      370797.473
#Sta/Elev= 30
       0 2371.14    20.1 2364.56    40.3 2350.99   100.7 2319.96   120.9 2304.14
   171.2 2278.14   191.4 2262.38   211.5 2255.22   312.2 2242.31   342.4 2236.06
   453.2 2220.46   503.6 2209.25   715.1 2196.18     716 2196.24     731 2197.45
   765.5  2200.3   785.6 2206.07   795.7 2215.28   856.1 2248.82   866.2 2256.04
   876.3 2267.35   936.7 2268.78  1017.3 2290.18  1027.4 2296.66  1087.8 2324.78
  1107.9 2337.43  1168.4  2360.4  1188.5 2371.94  1238.9 2392.97    1259 2405.09
#Mann= 3 , 0 , 0
       0      .1       0     716    .045       0     731      .1       0
Bank Sta=716,731
XS Rating Curve= 0 ,0
Exp/Cntr=0.3,0.1

Type RM Length L Ch R = 1 ,22289.6 ,814.5,800.6,786.7
XS GIS Cut Line= 2
     2224473.077      369973.074      2223314.07      370472.563
#Sta/Elev= 30
       0 2500.61    10.1 2489.08    80.8 2442.13     101 2423.34   161.5 2384.31
   191.8 2359.94   252.4 2320.41   262.5 2309.59   272.6 2302.58   333.2 2265.57
   353.4 2247.44     414 2205.74   434.2 2195.96   471.2 2193.67   486.2 2193.79
   646.2 2194.69   767.3 2192.21     838 2194.11   848.1 2196.55   858.2 2204.71
   928.9 2238.77   959.2 2257.54   979.4 2263.97  1019.7 2268.92  1090.4 2287.91
  1100.5 2291.69  1110.6 2298.74  1181.3 2324.74  1201.5 2335.18  1262.1 2358.49
#Mann= 3 , 0 , 0
       0      .1       0   471.2    .045       0   486.2      .1       0
Bank Sta=471.2,486.2
XS Rating Curve= 0 ,0
Exp/Cntr=0.3,0.1

Type RM Length L Ch R = 1 ,21489   ,772.2,773.1,773.9
XS GIS Cut Line= 2
     2223755.365      369134.128     2223076.449       370249.49
#Sta/Elev= 30
       0 2413.03      10 2410.36    50.2 2391.04    90.4 2366.41   110.5 2350.91
   130.6 2341.97   170.8 2313.86   210.9 2289.07   241.1 2272.96   261.2 2266.68
   341.5 2224.06   361.6 2215.99     452 2195.84   552.4 2182.44   555.4 2182.47
   570.4 2182.73   803.5 2188.08   863.8 2202.36     904  2218.6   964.2 2257.37
   974.3 2258.72   984.3 2263.64  1014.5 2281.46  1094.8 2323.09  1114.9 2327.99
  1205.3 2367.26  1225.4 2372.77  1255.5 2387.49  1285.6 2407.69  1305.7 2418.56
#Mann= 3 , 0 , 0
       0      .1       0   555.4    .045       0   570.4      .1       0
Bank Sta=555.4,570.4
XS Rating Curve= 0 ,0
Exp/Cntr=0.3,0.1

Type RM Length L Ch R = 1 ,20715.9 ,800.7,807.4,815.3
XS GIS Cut Line= 3
     2222867.925      368615.242     2222892.172      369182.622
     2222446.027      369837.291
#Sta/Elev= 30
       0 2331.42    29.9 2330.79    49.8 2324.74   109.6 2314.32   189.3 2292.74
   209.2 2289.98   288.9 2263.66   308.9 2260.59   388.6 2237.48   408.5 2234.23
   478.2 2214.19   498.2 2211.25   577.9 2187.88   678.2 2180.91   856.3 2176.44
   858.7 2176.42   871.3 2177.02  1029.2 2184.77  1039.2 2188.81  1099.4 2235.98
  1119.4 2243.15  1179.6 2288.14  1219.7 2325.57  1229.8 2330.97  1239.8 2333.18
  1259.8  2346.9  1279.9 2351.09  1340.1 2353.53  1350.1 2352.28  1360.1 2347.09
#Mann= 3 , 0 , 0
       0      .1       0   856.3    .045       0   871.3      .1       0
Bank Sta=856.3,871.3
XS Rating Curve= 0 ,0
Exp/Cntr=0.3,0.1

Type RM Length L Ch R = 1 ,19908.5 ,965.6,967.5,968.2
XS GIS Cut Line= 2
     2222572.111      368523.103     2221553.737      369366.899
#Sta/Elev= 30
       0  2321.5    40.4 2319.19     111 2296.02   131.2 2287.57   141.3 2280.08
   161.5 2271.26     212 2245.26   232.2 2237.46   242.3 2230.15   252.4 2224.96
   333.2 2194.97   363.4 2181.62     423 2168.01   434.1 2167.51     438 2167.54
   555.3  2169.6   666.3 2174.79   807.6 2173.07  1009.6 2173.25  1039.8 2174.52
    1050  2176.9  1080.2 2188.68  1120.6 2210.51    1161 2229.22  1181.2 2240.61
  1231.7 2260.46  1251.9 2264.98    1262 2268.95  1282.1 2281.73  1322.5 2301.26
#Mann= 3 , 0 , 0
       0      .1       0     423    .045       0     438      .1       0
Bank Sta=423,438
XS Rating Curve= 0 ,0
Exp/Cntr=0.3,0.1

Type RM Length L Ch R = 1 ,18941   ,752.2,748.5,744.7
XS GIS Cut Line= 2
       2222256.9      367955.723     2221073.646      368741.326
#Sta/Elev= 30
       0 2311.41    30.2  2299.7    40.3 2293.34    60.4 2287.43   120.9  2263.6
     141 2252.98   161.2 2245.39   191.4    2227   221.6 2212.97   241.8 2201.25
   332.4 2174.26   372.7 2165.78   392.8 2163.33   657.2 2160.35   672.2 2160.23
   674.9 2160.22     967 2164.33   987.2 2165.81  1077.8 2185.34    1098 2193.82
  1158.4    2215  1178.6 2222.77  1198.7 2235.22  1228.9 2247.84  1259.1 2265.42
  1289.4 2279.55  1299.4 2279.49  1369.9 2266.13  1400.2 2265.63  1420.3 2268.73
#Mann= 3 , 0 , 0
       0      .1       0   657.2    .045       0   672.2      .1       0
Bank Sta=657.2,672.2
XS Rating Curve= 0 ,0
Exp/Cntr=0.3,0.1

Type RM Length L Ch R = 1 ,18192.4 ,708.8,712.7,716.6
XS GIS Cut Line= 2
     2221985.333      367310.753     2220782.682      368169.097
#Sta/Elev= 30
       0 2329.12      10 2323.52    20.1  2314.5   100.5 2272.56   120.6 2259.06
   221.1 2216.73   261.3 2204.46   321.6 2190.68     402 2182.11   512.6 2162.31
   572.9  2156.2   663.4 2152.58   670.3 2152.78   685.3 2153.72   713.6 2157.14
   763.9 2159.17  1035.3 2162.61  1055.4 2172.38  1085.5 2192.54  1105.6 2211.26
  1145.8 2237.39    1186 2259.49  1196.1 2270.15  1206.2 2277.64  1236.3 2295.69
  1296.6 2315.72    1367 2329.84  1397.1 2339.73  1457.4 2354.21  1477.5  2362.8
#Mann= 3 , 0 , 0
       0      .1       0   670.3    .045       0   685.3      .1       0
Bank Sta=670.3,685.3
XS Rating Curve= 0 ,0
Exp/Cntr=0.3,0.1

Type RM Length L Ch R = 1 ,17479.7 ,804.1,807.2,810.3
XS GIS Cut Line= 2
     2221611.245      366831.316     2220427.067      367510.245
#Sta/Elev= 30
       0 2259.97    50.2 2237.31    70.3 2224.53    90.3 2217.43   140.5 2208.55
   160.6 2201.31   240.9 2180.74   250.9 2175.78   321.2  2158.8   341.2 2151.82
   592.2  2150.5     675 2145.89   682.5 2145.63     690 2145.76   893.3 2150.54
   943.5 2154.26   953.5  2158.4   973.6 2175.56   993.6 2185.19  1053.9 2222.73
  1073.9    2240  1144.2 2282.46  1164.3 2298.43  1194.4 2316.15  1214.4  2323.7
  1234.5 2334.45  1284.7 2332.83  1314.8 2341.35  1344.9  2353.2    1365 2352.72
#Mann= 3 , 0 , 0
       0      .1       0     675    .045       0     690      .1       0
Bank Sta=675,690
XS Rating Curve= 0 ,0
Exp/Cntr=0.3,0.1

Type RM Length L Ch R = 1 ,16672.5 ,791.7,792.3,792.8
XS GIS Cut Line= 2
     2221408.255      366142.047     2220103.765      366714.276
#Sta/Elev= 30
       0 2270.28   100.3 2242.12   160.5 2231.35   220.7 2212.93   351.1  2183.9
   401.3 2169.33   431.4 2164.57   531.7  2140.9   672.1  2140.5   832.6 2136.29
   846.1 2136.73   861.1  2138.6   882.8  2142.1     953 2143.02     963 2145.96
  1023.2 2178.72  1033.2 2185.76  1043.3 2196.79  1113.5 2243.54  1133.6 2264.34
  1203.8 2310.12  1223.8 2329.66  1253.9 2348.92  1294.1 2367.89  1304.1 2376.12
  1324.2 2386.22  1374.3 2403.35  1384.4 2410.54  1414.4 2419.58  1424.5  2419.5
#Mann= 3 , 0 , 0
       0      .1       0   846.1    .045       0   861.1      .1       0
Bank Sta=846.1,861.1
XS Rating Curve= 0 ,0
Exp/Cntr=0.3,0.1

Type RM Length L Ch R = 1 ,15880.3 ,1054.6,1048.7,1042.7
XS GIS Cut Line= 2
     2221002.473       365476.82     2219740.448      365996.934
#Sta/Elev= 30
       0 2249.14    20.1 2226.11    30.1 2219.41    50.2 2209.26    90.3 2194.68
   100.4 2188.74   180.7 2167.28   190.7 2162.69   250.9 2147.47     271 2140.05
   291.1 2138.94   331.2 2141.47     552 2137.86   688.4 2131.98   692.5 2131.75
   703.4 2131.95   792.9  2136.6   853.1  2156.1   893.3 2162.92   913.4 2168.58
   933.4 2176.93   973.6 2201.31  1013.7 2228.78  1033.8 2246.81    1104 2289.97
  1114.1 2293.46  1184.3 2305.78  1264.6 2329.77  1344.9 2360.87    1365 2372.99
#Mann= 3 , 0 , 0
       0      .1       0   688.4    .045       0   703.4      .1       0
#XS Ineff= 2 , 0
          330.65  2141.3
Permanent Ineff=
       F       F
Bank Sta=688.4,703.4
XS Rating Curve= 0 ,0
Exp/Cntr=0.3,0.1

Type RM Length L Ch R = 1 ,14831.6 ,535.3,534.8,534.2
XS GIS Cut Line= 2
     2220617.802      364367.166     2219483.042      365235.209
#Sta/Elev= 30
       0 2311.16    10.1 2310.11    70.4 2285.46   110.7 2265.53   201.2 2224.61
   241.5 2203.78   281.7 2187.26   291.8 2182.12   352.1 2162.49   382.3 2155.32
   402.4 2147.13   442.7 2135.03   600.5 2123.24   603.7 2122.97   615.5 2123.33
   724.4 2128.19   935.7 2129.63  1106.7 2132.42  1126.9 2133.96  1136.9 2137.03
  1177.2 2155.36  1187.2 2160.63  1197.3 2168.32  1267.7 2208.83  1277.8 2213.94
  1287.8 2217.42    1308 2231.53  1388.4 2279.67  1398.5 2289.66  1428.7 2311.87
#Mann= 3 , 0 , 0
       0      .1       0   600.5    .045       0   615.5      .1       0
Bank Sta=600.5,615.5
XS Rating Curve= 0 ,0
Exp/Cntr=0.3,0.1

Type RM Length L Ch R = 1 ,14296.9 ,311.6,309.9,308.1
XS GIS Cut Line= 2
     2220369.311      364009.795     2219248.957      364789.558
#Sta/Elev= 30
       0    2407      10 2400.52    20.1  2391.1   100.4  2341.8   120.4 2324.99
   160.6 2300.78   180.7 2289.59   200.7 2281.64   220.8 2266.42   301.1 2223.43
   311.1 2215.77   341.2  2198.6   351.3 2191.25   381.4  2179.4   401.5  2169.4
   411.5 2162.05   421.5 2156.88   501.8 2120.15   511.9 2117.26   632.3 2114.54
   638.7 2114.55   653.7 2114.74   953.5 2119.16    1084 2123.53  1174.3 2138.69
  1254.6 2154.94  1264.6 2158.78  1274.7 2165.83  1334.9 2195.99    1365 2214.67
#Mann= 3 , 0 , 0
       0      .1       0   638.7    .045       0   653.7      .1       0
Bank Sta=638.7,653.7
XS Rating Curve= 0 ,0
Exp/Cntr=0.3,0.1

Type RM Length L Ch R = 1 ,13986.9 ,749.8,751.6,753.4
XS GIS Cut Line= 2
     2220001.928      363862.828     2219109.638      364629.034
#Sta/Elev= 30
       0 2242.93    20.1 2239.54    70.4 2235.82    90.5 2227.13   110.6 2214.75
   120.6 2205.83   180.9 2179.05   211.1 2163.86   231.2 2149.26   241.2 2144.59
   281.5 2130.56   351.4 2113.26   361.9 2112.34   366.4 2112.42   452.4 2116.25
   522.7  2117.5   794.1 2117.77   884.6 2120.46   934.9 2137.07   985.1 2146.64
   995.2 2152.25  1015.3 2169.22  1025.3 2174.45  1055.5  2186.7  1065.5 2194.31
  1075.6 2199.42  1105.8 2212.87    1156 2232.38  1166.1 2238.72  1176.1 2246.73
#Mann= 3 , 0 , 0
       0      .1       0   351.4    .045       0   366.4      .1       0
Bank Sta=351.4,366.4
XS Rating Curve= 0 ,0
Exp/Cntr=0.3,0.1

Type RM Length L Ch R = 1 ,13235.2 ,724,722.3,720.6
XS GIS Cut Line= 2
     2219565.482      363295.448     2218653.794      364139.244
#Sta/Elev= 30
       0 2262.85    70.1 2230.19    90.2 2218.88   130.2 2202.68   150.3  2196.5
   170.3 2187.75   180.3  2182.7   190.3 2174.92   200.4 2169.55   260.5 2142.21
   300.5 2119.48   330.6 2114.22   340.6 2114.07   380.7 2118.78   420.8 2116.89
   520.9 2108.44   631.1 2107.56   674.1 2107.63   689.1 2107.57   881.6 2112.17
   891.6 2113.47   951.7 2137.76   961.7 2145.74   971.8 2151.09  1021.8 2174.15
  1051.9 2185.77  1071.9 2196.62    1112 2206.02  1142.1 2216.23  1242.2 2258.41
#Mann= 3 , 0 , 0
       0      .1       0   674.1    .045       0   689.1      .1       0
Bank Sta=674.1,689.1
XS Rating Curve= 0 ,0
Exp/Cntr=0.3,0.1

Type RM Length L Ch R = 1 ,12513   ,469.2,473.7,478.3
XS GIS Cut Line= 2
     2219182.379      362762.014     2218222.198      363586.412
#Sta/Elev= 30
       0 2196.83    70.3 2169.13   110.5  2158.5   180.8 2146.11   200.9 2141.66
   210.9 2136.82   261.1 2118.52   291.3 2113.75   321.4 2111.38   441.9 2106.47
   522.3 2107.32     693 2106.73   743.2 2108.06   783.4 2106.83   825.3  2104.2
   833.6 2103.59   840.3 2103.92   843.7 2104.09   863.8 2109.82     914 2112.24
     924 2114.44   954.2 2124.19  1044.6 2166.86  1094.8 2197.04  1104.8 2199.42
  1114.9 2203.18    1155 2228.48  1175.1 2244.22  1185.2 2250.03  1265.5 2289.78
#Mann= 3 , 0 , 0
       0      .1       0   825.3    .045       0   840.3      .1       0
Bank Sta=825.3,840.3
XS Rating Curve= 0 ,0
Exp/Cntr=0.3,0.1

Type RM Length L Ch R = 1 ,12039.3 ,326.7,328.5,330.3
XS GIS Cut Line= 3
     2218989.867      362657.635     2218355.507      363041.388
     2218135.409      363504.663
#Sta/Elev= 30
       0 2169.55      20 2161.39    40.1 2150.53   100.2 2130.16   130.2 2117.34
   150.3 2111.94   310.6  2104.6   400.8 2102.28   435.2 2102.53   450.2  2103.8
     501 2107.76   661.2 2107.56   791.7 2112.44   821.9 2111.48     842 2113.46
   922.4  2113.2   972.7 2118.22  1043.1  2133.3  1053.2  2137.8  1083.3 2164.43
  1093.4 2171.25  1123.6 2186.26  1133.6 2190.26  1143.7 2188.95  1183.9 2209.02
    1194 2212.76  1214.1 2217.27  1224.1 2222.24  1244.2 2226.25  1254.3 2224.68
#Mann= 3 , 0 , 0
       0      .1       0   435.2    .045       0   450.2      .1       0
Bank Sta=435.2,450.2
XS Rating Curve= 0 ,0
Exp/Cntr=0.3,0.1

Type RM Length L Ch R = 1 ,11710.7 ,436.3,433,429.2
XS GIS Cut Line= 3
     2218857.208      362409.617     2217969.011      362851.857
     2217523.055      363093.417
#Sta/Elev= 30
       0 2184.82      20 2174.99    30.1 2167.01    40.1 2161.81   100.2  2137.4
   110.2 2131.02   170.4 2111.55   200.4 2107.64   370.8 2100.34   383.3 2101.59
   398.3 2102.81   691.5 2104.16   972.2 2112.06    1022 2113.96  1041.9  2116.5
  1071.8 2125.44  1081.7 2131.02  1091.6 2134.26  1161.3 2154.89    1211  2175.5
  1240.8 2189.91  1260.7  2204.5  1300.5 2228.25  1330.3 2247.95  1350.2 2266.97
  1399.9 2299.82  1429.8 2322.75  1439.7 2335.04  1459.6 2345.14  1499.4 2356.15
#Mann= 3 , 0 , 0
       0      .1       0   383.3    .045       0   398.3      .1       0
Bank Sta=383.3,398.3
XS Rating Curve= 0 ,0
Exp/Cntr=0.3,0.1

Type RM Length L Ch R = 1 ,11277.7 ,544.4,535.1,526.3
XS GIS Cut Line= 3
     2218481.861      362145.759     2217894.685      362550.836
     2217485.256      362952.321
#Sta/Elev= 30
       0 2151.02      10 2144.72    40.2 2131.32    80.4 2115.66    90.4 2113.53
   110.5 2110.41   261.2  2104.7   328.5 2099.77   331.6 2099.66   343.5 2100.09
   371.7 2101.97   512.4 2101.17   592.8 2103.66   693.2 2104.88     824 2110.35
   884.4 2110.11   894.4 2111.78   924.6 2120.76   934.7 2124.86   974.9 2146.32
     995 2154.95  1005.1 2160.35  1045.3 2187.05  1115.8 2227.59  1135.9 2244.79
    1156 2253.32  1206.3  2284.6  1226.4 2297.37  1246.5 2313.61  1286.8 2338.69
#Mann= 3 , 0 , 0
       0      .1       0   328.5    .045       0   343.5      .1       0
Bank Sta=328.5,343.5
XS Rating Curve= 0 ,0
Exp/Cntr=0.3,0.1

Type RM Length L Ch R = 1 ,10742.6 ,461.4,479.6,497.8
XS GIS Cut Line= 3
     2218484.065       361738.79     2217906.986      361879.423
     2217320.209      362737.767
#Sta/Elev= 30
       0 2331.53    40.3 2307.31    50.3    2297   120.8 2259.02   140.9 2244.06
   191.3 2218.08   211.4  2203.6   271.8 2175.63     292 2163.66   372.5 2134.69
     453 2113.79   473.2 2110.66   553.7 2105.92   694.9 2102.38   748.6  2094.5
   763.6 2094.75     806 2098.27   896.8  2088.4  1038.1 2100.12  1179.4 2102.44
  1219.8 2106.94  1270.3 2118.73  1320.8 2132.69    1341 2141.07  1421.7 2182.07
  1441.9 2186.88  1542.9 2236.08  1573.1 2245.37  1593.3 2254.17  1633.7 2275.54
#Mann= 3 , 0 , 0
       0      .1       0   748.6    .045       0   763.6      .1       0
Bank Sta=748.6,763.6
XS Rating Curve= 0 ,0
Exp/Cntr=0.3,0.1

Type RM Length L Ch R = 1 ,10263   ,802.1,796.9,791.7
XS GIS Cut Line= 2
     2218212.499      361539.965     2216874.064      361777.585
#Sta/Elev= 30
       0 2216.58    50.4 2190.09    60.4  2180.9     141 2137.95   161.1 2131.28
   191.3 2124.36   231.6 2116.71   342.4 2103.75   392.7 2100.65   523.6 2097.25
   654.5 2088.77   701.1  2090.2   716.1 2090.66   775.3 2095.08   956.6 2094.55
  1027.1 2100.58  1047.2 2107.92  1057.3 2113.17  1067.4 2120.98  1077.4 2140.52
  1087.5 2150.06  1097.6 2155.72  1127.8  2164.7  1147.9 2172.98  1198.2 2175.33
  1218.4 2179.63  1238.5 2191.21  1288.9 2210.96    1309 2223.54  1359.4 2244.47
#Mann= 3 , 0 , 0
       0      .1       0   701.1    .045       0   716.1      .1       0
#XS Ineff= 2 , 0
                          856.85         2095.58
Permanent Ineff=
       F       F
Bank Sta=701.1,716.1
XS Rating Curve= 0 ,0
Exp/Cntr=0.3,0.1

Type RM Length L Ch R = 1 ,9466    ,769.3,779,788.6
XS GIS Cut Line= 2
     2218357.981      360502.193     2216752.829      361205.356
#Sta/Elev= 30
       0  2214.4    60.4 2194.41    90.6 2188.76   151.1 2169.48   292.1 2138.84
   322.3 2136.13   382.7 2123.63     423 2110.66   503.6 2092.44   543.8 2088.81
   866.1 2087.03   916.5 2083.37  1057.5  2082.4  1067.6 2082.27  1072.5 2082.35
  1168.3 2084.08  1188.4 2087.16  1238.8  2108.8  1258.9 2121.32  1319.4 2145.29
  1339.5 2158.24    1410 2191.03  1430.1 2206.48  1490.6 2238.97  1510.7 2257.09
  1581.2 2303.61  1591.3 2315.74  1661.8  2359.9  1681.9 2376.42  1752.4 2412.02
#Mann= 3 , 0 , 0
       0      .1       0  1057.5    .045       0  1072.5      .1       0
Bank Sta=1057.5,1072.5
XS Rating Curve= 0 ,0
Exp/Cntr=0.3,0.1

Type RM Length L Ch R = 1 ,8687    ,643.6,642.7,641.8
XS GIS Cut Line= 2
     2218132.024       360173.03     2216645.064      360185.634
#Sta/Elev= 30
       0 2176.06    20.1 2170.36    30.1 2165.47   120.6 2140.14   160.8 2126.21
   170.8 2119.03     211 2096.32   231.1 2090.07   321.5 2084.56   411.9 2081.67
   773.6 2075.81   823.9 2078.43   864.1 2074.56   871.1  2074.7   886.1 2074.98
   914.3 2075.96   934.4 2081.51   994.7 2090.57  1085.1 2109.19  1145.4 2118.78
  1175.5 2126.44  1215.7 2143.22  1235.8 2155.94  1296.1 2182.37  1316.2 2195.84
  1366.4 2218.07  1386.5 2231.79  1436.8 2255.59  1456.9 2268.32    1487 2281.17
#Mann= 3 , 0 , 0
       0      .1       0   871.1    .045       0   886.1      .1       0
Bank Sta=871.1,886.1
XS Rating Curve= 0 ,0
Exp/Cntr=0.3,0.1
